HEC-RAS study NFSBPOTOMC.prj: NFSBPOTOMC

--- NFSBPOTOMC.g01 (geometry) --- (continued)

Type RM Length L Ch R = 1 ,62632   ,546.6,535.3,523.8
XS GIS Cut Line= 3
2425918.31418943663636.7832932172426687.38286129663534.610925376
2428041.58192453663323.822304964
#Sta/Elev= 30
       0 1646.77   221.7 1625.67   247.8 1626.36     291 1621.91   319.2 1622.94
   383.8 1616.82   399.9 1613.82   416.1 1605.41   428.2 1594.17   432.2 1592.07
   444.3 1588.59     521 1588.59   545.2 1591.87   557.3  1595.6   569.4 1602.96
   577.5 1604.57   597.6 1604.21   617.2 1599.82   714.5 1603.82     844 1599.75
   916.9 1602.05   978.2 1600.91  1101.4 1604.56  1418.8  1605.4  1685.8 1604.76
    1910 1601.63    1945 1603.68  1977.5 1620.87    2107 1718.57  2146.3 1750.16
#Mann= 10 ,-1 , 0
       0     .05       0   221.7     .06       0   319.2    .055       0
   432.2    .045       0   545.2    .055       0   617.2     .06       0
   714.5     .05       0   916.9     .05       0  1418.8     .05       0
    1910      .1       0
#XS Ineff= 2 ,-1
  907.08 1353.98  1606.8 1353.98  2053.1  1611.9
Permanent Ineff=
       F       F
Bank Sta=432.2,545.2
XS Rating Curve= 0 ,0
Exp/Cntr=0.5,0.3

Type RM Length L Ch R = 1 ,62097   ,664.6,657.3,637.4
XS GIS Cut Line= 3
2426031.77787328664244.5406078852426673.04430726 664046.54756555
2428182.27980587663589.111472547
#Sta/Elev= 30
       0 1684.41    78.5 1678.75   141.3 1669.03   290.3 1664.47   325.5 1661.75
   346.4 1653.94   388.2 1653.85   413.4 1651.69   421.7 1646.29   450.2 1618.45
   467.41594.885   476.2 1588.32   480.3 1586.97   580.8 1586.67   619.21594.327
   821.6 1601.46   936.2  1600.9  1074.2  1597.7    1148  1601.2  1776.4 1599.16
  1985.3 1596.54  2051.5 1598.26  2068.9 1603.72  2095.6 1618.24  2144.2 1654.29
  2160.9 1669.22  2177.6 1690.35    2199 1712.32  2218.2 1728.79  2248.2 1748.45
#Mann= 8 ,-1 , 0
       0     .05       0  303.89     .06       0  404.17      .1       0
   467.4    .045       0   619.2    .055       0  704.98     .05       0
 1105.82     .05       0  2007.7      .1       0
#XS Ineff= 1 ,-1
 1176.99 2248.17 1607.34
Permanent Ineff=
       F
Bank Sta=467.4,619.2
XS Rating Curve= 0 ,0
Exp/Cntr=0.3,0.1

Type RM Length L Ch R = 1 ,61439   ,582.3,579.9,580.3
XS GIS Cut Line= 3
2426285.13268152664951.8105188012427064.35750103664543.355298966
2428397.77740636663952.861073121
#Sta/Elev= 30
       0 1720.82    83.1 1709.26   158.9 1684.16   194.5 1684.85   340.5 1669.26
   394.7 1660.43   421.8 1659.19   439.9 1647.11   471.5 1646.56   485.1 1651.37
   585.6 1634.49   594.5  1629.7  639.851589.759   650.8 1586.15   694.5 1583.51
   774.1 1583.47  791.811589.509   841.8 1597.99   861.2 1590.58   899.9 1589.47
  1021.4 1597.13  1394.2 1594.28  1709.7 1596.32  1809.5 1592.75  2151.1 1592.34
  2172.9 1602.11  2225.1 1637.97    2291 1707.79  2330.4 1739.09  2338.1  1741.3
#Mann= 10 ,-1 , 0
       0      .1       0  382.37     .06       0  487.07      .1       0
  639.85    .045       0  791.81      .1       0  905.36     .05       0
 1521.35     .06       0 1726.68     .05       0 1829.34      .1       0
 2137.34      .1       0
#XS Ineff= 2 , 0
                         1216.81         1602.78
Permanent Ineff=
       F       F
Bank Sta=639.85,791.81
XS Rating Curve= 0 ,0
Exp/Cntr=0.3,0.1

Type RM Length L Ch R = 1 ,60859   ,424.6,421.5,419.9
XS GIS Cut Line= 2
2426743.29022977665341.1830996272428580.86627904664441.965081796
#Sta/Elev= 30
       0  1654.4   186.4 1629.45   253.2 1617.34   293.3 1616.78   333.2 1610.54
   351.2 1611.34   377.9 1603.34   462.5 1597.42   496.6 1586.06  519.44 1584.26
   542.7 1581.34   627.3 1581.34  639.311585.952   645.1 1588.71     689 1596.23
   721.9 1589.62   822.3 1590.26   933.4 1585.91   961.3 1590.97    1161 1588.29
  1246.3 1590.64  1358.8 1588.81  1451.2  1591.4  1869.8 1588.76  1926.9 1597.22
  1941.9 1602.95  1977.7 1626.71  2012.3 1655.57  2028.6 1663.08  2045.8 1682.59
#Mann= 11 ,-1 , 0
       0      .1       0  179.11     .06       0  282.89    .055       0
  354.41      .1       0  386.67     .05       0  519.44    .045       0
  639.31    .025       0  683.45    .055       0  698.01     .05       0
 1735.81      .1       0 1943.37      .1       0
#XS Ineff= 2 , 0
                         1442.48         1597.79
Permanent Ineff=
       F       F
Bank Sta=519.44,639.31
XS Rating Curve= 0 ,0
Exp/Cntr=0.3,0.1

Type RM Length L Ch R = 1 ,60438   ,782.8,766.9,744.6
XS GIS Cut Line= 3
2427019.75063485665692.8966350412427597.67730051665385.364441708
 2428834.2283051664880.116764545
#Sta/Elev= 30
       0 1656.68    12.5 1651.22    30.6 1637.58    44.2 1634.62    63.9 1623.29
    80.4 1619.68   202.8 1617.64     261  1613.8   402.1 1613.08   411.2 1609.53
   442.9 1585.58   453.2 1582.95  476.841582.056   497.3 1580.28   578.8 1580.31
   586.81583.003   592.4 1588.37   598.1 1590.86   627.7 1586.28   841.4 1588.72
     866  1591.6   884.8 1589.19  1168.8 1586.42  1342.9 1587.64  1540.8 1584.58
  1809.5 1585.94  1844.1 1596.25  1891.6 1633.18  1923.4  1669.2  1990.4 1721.05
#Mann= 9 ,-1 , 0
       0      .1       0  162.08    .055       0     267    .035       0
  319.17      .1       0  371.92     .05       0  476.84    .045       0
   586.8      .1       0  685.77     .05       0 1807.05      .1       0
Bank Sta=476.84,586.8
XS Rating Curve= 0 ,0
Exp/Cntr=0.3,0.1

Type RM Length L Ch R = 1 ,59671   ,691.2,701.1,696.6
XS GIS Cut Line= 4
2427661.56332761666267.5404988832427942.37346151666081.087787792
2428442.33473194 665494.496441292428971.19522277  665268.6425623
#Sta/Elev= 30
       0 1659.17    90.8 1647.79   102.2 1645.04   131.2 1645.27   145.6 1641.08
   303.9 1622.92     340 1614.31   381.5 1599.87     424 1582.78   492.4 1584.44
   504.8  1581.2   520.5 1576.96   634.3 1576.77   639.7 1577.02  648.571581.779
   665.8 1584.15   798.6 1582.84   837.1 1587.19  1065.3 1586.06  1110.9 1582.93
    1437 1584.28  1510.2 1581.09  1534.5 1587.98  1573.7 1613.22  1582.4 1625.39
  1591.1 1632.85  1599.8 1644.57  1612.8 1656.91  1630.2 1676.29  1682.9 1721.44
#Mann= 7 ,-1 , 0
       0      .1       0   10.01     .06       0  211.39      .1       0
   504.8    .045       0  648.57      .1       0   854.4     .05       0
  1525.9      .1       0
Bank Sta=504.8,648.57
XS Rating Curve= 0 ,0
Exp/Cntr=0.3,0.1

Type RM Length L Ch R = 1 ,58970   ,477.2,481.5,489.6
XS GIS Cut Line= 4
2428012.56164137666841.8290484552428328.92846268666603.862660885
2428968.24345702665989.1368562132429143.01377678665918.168166131
#Sta/Elev= 30
       0 1649.31    51.5 1645.42    84.7 1638.53   142.9 1638.16   186.5 1630.58
   386.4 1614.93   397.3 1610.57   431.8 1585.24   457.3 1578.68   478.1 1581.29
   814.6 1578.66   830.7 1581.04  847.321574.977     859 1571.72   945.5 1569.97
  959.181576.902   969.3 1581.14  1147.5 1579.37  1164.5 1581.88  1199.5  1595.9
    1272 1633.81  1275.2 1637.29  1285.5 1657.98  1298.4 1669.47  1311.4 1699.15
  1315.7 1704.25  1335.6 1713.82  1350.2 1727.17  1433.8 1781.33  1471.4 1797.33
#Mann= 8 ,-1 , 0
       0     .05       0   59.32     .06       0  171.54     .05       0
  395.97      .1       0  516.72     .05       0  847.32    .045       0
  959.18     .05       0  967.48      .1       0
Bank Sta=847.32,959.18
XS Rating Curve= 0 ,0
Exp/Cntr=0.3,0.1

Type RM Length L Ch R = 1 ,58488   ,481.9,491.9,506.5
XS GIS Cut Line= 3
2428167.23652884667208.938550457 2428474.7844702666979.511187792
2429194.86833185666470.263518631
#Sta/Elev= 30
       0 1665.24    36.9  1660.5    75.4 1651.62   130.5 1650.84   164.1 1646.73
   218.3 1631.82   248.9 1628.07   317.8 1627.49   343.7 1630.23   403.2 1622.52
   457.1 1593.09   481.8 1589.64   507.5 1576.31   530.6 1572.32   555.1 1575.09
     648 1578.06   772.7 1575.79   943.7 1576.33   958.1 1581.08   986.8 1571.31
 1038.181570.001  1058.5 1567.58  1118.5 1567.59 1129.971572.059  1147.5 1583.68
  1187.1 1618.24  1202.2 1640.87  1222.1 1658.61    1241 1682.73  1265.7 1708.57
#Mann= 13 ,-1 , 0
       0     .06       0   50.18     .05       0   65.28     .06       0
  177.26     .05       0  289.24      .1       0     401      .1       0
  471.43      .1       0  511.55     .05       0  843.21      .1       0
   909.6    .025       0  953.77     .05       0 1038.18    .045       0
 1129.97      .1       0
Bank Sta=1038.18,1129.97
XS Rating Curve= 0 ,0
Exp/Cntr=0.3,0.1

Type RM Length L Ch R = 1 ,57997   ,471.4,468,461.3
XS GIS Cut Line= 3
2428177.03178486667408.7655786282428583.12677318667259.060169384
2429364.51989543666985.195887715
#Sta/Elev= 30
       0 1668.51    55.7 1657.43   116.9 1650.71   129.7 1646.59   167.9 1646.78
   180.9 1642.05   219.2 1637.98   240.6 1632.04   300.2 1631.45     377 1628.05
   457.8 1621.33   474.8 1613.91   525.7 1581.13   559.6 1569.88   611.5 1573.49
   682.5 1573.89   746.5 1576.56   949.5 1573.67   979.2 1574.05   996.1 1576.48
  1013.1 1568.09 1032.811566.832    1047    1564  1123.3 1564.01 1140.811567.946
  1160.8 1573.48  1174.2 1582.19  1208.1 1613.84  1246.2  1654.3  1260.8 1666.81
#Mann= 7 ,-1 , 0
       0      .1       0   81.71     .06       0   182.9     .05       0
   990.7      .1       0 1032.81    .045       0 1140.81      .1       0
 1184.98      .1       0
Bank Sta=1032.81,1140.81
XS Rating Curve= 0 ,0
Exp/Cntr=0.3,0.1

Type RM Length L Ch R = 1 ,57529   ,369.3,368.9,369.7
XS GIS Cut Line= 2
2428342.06295085667940.9862989632429623.27364302667358.326046959
#Sta/Elev= 30
       0 1677.78    62.3 1662.01   119.4 1629.75   145.8 1609.69   176.5  1609.5
   211.7 1600.55   273.9 1591.93   435.8 1588.68   475.3 1578.85   576.4  1570.9
   615.9 1572.34   686.2 1568.44   769.7 1573.06  1056.3  1569.2  1094.9 1575.67
 1115.591567.759  1122.7 1563.52  1134.5 1562.28    1174 1562.43 1195.561565.646
  1234.5 1564.97  1253.1 1568.78  1266.3  1575.6  1294.9 1602.53  1310.2 1623.91
  1319.2 1632.43  1334.2 1654.86    1341 1672.26  1345.4 1678.37  1407.5 1726.45
#Mann= 6 ,-1 , 0
       0      .1       0  105.51     .06       0  208.45     .05       0
 1115.59    .045       0 1195.56      .1       0 1237.83      .1       0
Bank Sta=1115.59,1195.56
XS Rating Curve= 0 ,0
Exp/Cntr=0.3,0.1

Type RM Length L Ch R = 1 ,57160   ,386.7,385.3,384.5
XS GIS Cut Line= 2
2428422.19664887668354.6396711322429791.80841094667673.572135627
#Sta/Elev= 30
       0 1712.29    40.8 1706.32      81 1692.59   130.2 1665.41   155.4 1648.62
   161.4 1642.82   174.8 1624.29   197.1 1603.52   237.4 1602.06     242 1600.77
   259.7 1589.66   268.6 1587.68   509.9 1573.82   715.4 1573.87   834.9 1569.17
   934.3 1568.62   987.6 1566.38  1122.1 1566.25  1193.7 1569.64  1226.5 1574.91
  1251.4 1573.49 1262.021566.224  1274.2 1560.75  1349.7 1560.03  1357.8 1561.96
 1365.861567.821  1376.5 1580.85  1418.8 1621.43  1461.4 1656.02  1529.6 1708.15
#Mann= 5 ,-1 , 0
       0      .1       0  197.06     .06       0  301.04     .05       0
 1262.02    .045       0 1365.86      .1       0
Bank Sta=1262.02,1365.86
XS Rating Curve= 0 ,0
Exp/Cntr=0.3,0.1

Type RM Length L Ch R = 1 ,56774   ,378.3,378.6,379
XS GIS Cut Line= 2
2428598.70974728668713.4214338812430038.66520068667977.060373798
#Sta/Elev= 30
       0    1709    37.6 1685.75   121.3 1627.95   161.8 1604.92   174.3 1595.52
     210 1592.93   230.8    1585   299.2 1573.18   399.9 1571.12   593.4 1571.56
   652.9 1569.45   772.8 1570.78   875.8 1567.91   997.4 1566.94  1158.2 1568.48
  1177.1 1563.99  1199.6 1562.41 1241.941565.143    1258 1561.89  1280.1 1560.01
  1352.3    1560  1361.3 1560.74  1365.8 1562.62 1369.731565.806  1416.8 1609.18
    1447 1633.84  1467.4 1647.35  1487.1 1662.91  1544.7 1704.45  1617.3 1759.46
#Mann= 5 ,-1 , 0
       0      .1       0   75.02     .06       0  283.72     .05       0
 1241.94    .045       0 1369.73      .1       0
Bank Sta=1241.94,1369.73
XS Rating Curve= 0 ,0
Exp/Cntr=0.3,0.1

Type RM Length L Ch R = 1 ,56396   ,338.1,342.8,349.6
XS GIS Cut Line= 3
2428784.46298468669037.627150297 2429938.3425667668453.498725384
 2430304.2017431668269.549290121
#Sta/Elev= 30
       0 1711.61    51.9 1686.52    85.8 1668.05   176.4 1613.01   226.7 1585.43
   256.7 1583.72   386.9 1569.36   519.7  1569.9   625.7 1566.21   813.3 1566.22
   869.9 1563.21  1136.8 1568.61  1204.1 1566.83 1217.471563.631    1233 1558.05
  1329.6 1556.57  1334.1 1557.31 1344.991563.935  1355.1  1571.6  1379.3 1582.73
  1408.8 1603.02  1454.9 1636.67  1492.2 1669.84  1530.6 1697.12  1548.4 1708.15
  1580.3 1723.35  1625.1 1734.52  1655.3 1746.49  1673.1 1750.76  1702.8 1761.74
#Mann= 6 ,-1 , 0
       0      .1       0  145.39     .06       0  770.69     .05       0
 1217.47    .045       0 1344.99      .1       0  1395.9      .1       0
Bank Sta=1217.47,1344.99
XS Rating Curve= 0 ,0
Exp/Cntr=0.5,0.3

Type RM Length L Ch R = 1 ,56053   ,54.4,51.7,50
XS GIS Cut Line= 2
2429030.55337179669119.7319729632430517.91883537668610.015800789
#Sta/Elev= 30
       0 1627.89    46.7 1600.52    80.5    1584    93.2 1583.71   113.6 1578.52
     152 1578.97   169.3 1574.73   241.2 1573.05   270.8 1566.16   350.4 1566.43
   376.5 1563.15   422.1 1562.81   815.9 1566.31   892.4 1564.57  1023.5 1566.81
  1078.4  1566.3 1089.421559.962  1103.8 1554.74  1167.2 1554.56 1193.18 1560.92
  1213.2 1572.15  1230.7  1576.1  1298.1 1606.48  1329.8 1616.05  1382.9 1647.82
    1404  1663.1  1414.2 1668.66  1467.4 1694.28  1522.4 1714.17  1572.3 1736.67
#Mann= 10 ,-1 , 0
       0      .1       0    8.21     .06       0  209.73     .05       0
  310.49    .055       0  411.24     .06       0  533.44     .05       0
  814.28     .06       0  1015.8    .055       0 1089.42    .045       0
 1193.18      .1       0
#XS Ineff= 2 ,-1
       0 1069.42  1565.5 1213.18 1572.28  1565.5
Permanent Ineff=
       F       F
Bank Sta=1089.42,1193.18
XS Rating Curve= 0 ,0
Exp/Cntr=0.5,0.3

Type RM Length L Ch R = 1 ,56001   ,357,347.6,337.1
XS GIS Cut Line= 2
2429076.67631102 669220.310840042430504.31157911668646.257526204
#Sta/Elev= 30
       0 1651.93      55 1614.45    88.5 1595.44   119.5 1581.13   153.1  1576.8
   200.5 1577.22   243.7 1571.56   282.5 1569.13     317 1561.65   405.5 1563.66
   531.6 1563.19   765.3 1565.94   842.9 1564.03  1071.4 1567.69    1080 1567.33
  1091.11560.324  1100.4 1555.48  1114.5 1554.56  1170.6 1554.59 1199.011560.802
  1226.6 1577.96  1281.8 1582.54  1301.1 1598.53  1354.8 1626.26    1400 1657.34
  1429.8 1669.41  1446.5 1679.37  1493.9 1701.35  1515.6 1708.81  1538.7 1719.29
#Mann= 8 ,-1 , 0
       0      .1       0   79.93     .06       0  385.35     .05       0
  452.43     .06       0  996.18    .055       0  1091.1    .045       0
 1199.01     .05       0 1199.79      .1       0
Bank Sta=1091.1,1199.01
XS Rating Curve= 0 ,0
Exp/Cntr=0.5,0.3

Type RM Length L Ch R = 1 ,55654   ,394.2,340.6,337.8
XS GIS Cut Line= 3
2429372.17342344669737.2766696212430100.93804201669228.166795462
 2430587.7369372 668919.15986754
#Sta/Elev= 30
       0 1711.37    32.1 1706.86    81.2 1696.53   125.1  1682.8   178.8 1653.94
   201.8  1637.5     213 1632.71   222.7 1623.48   236.2 1618.56   261.7 1601.83
   308.1 1579.85   325.2 1564.74   330.1 1563.38   356.9 1564.06   374.1 1558.54
   730.6 1564.32   863.3  1562.9  1050.6 1565.39 1087.811557.499  1104.3 1553.84
  1184.9 1554.29 1203.131558.219    1218 1563.23  1233.2 1574.91  1255.9 1596.92
    1268 1603.61    1381 1615.61  1398.1 1621.67  1440.7 1641.97  1465.6 1656.27
#Mann= 6 ,-1 , 0
       0      .1       0  295.59     .06       0  405.84     .05       0
 1063.76      .1       0 1087.81    .045       0 1203.13      .1       0
Bank Sta=1087.81,1203.13
XS Rating Curve= 0 ,0
Exp/Cntr=0.3,0.1

Type RM Length L Ch R = 1 ,55313   ,530.5,499.8,497.6
XS GIS Cut Line= 4
2429622.03906545670123.2867243742429877.09301728669919.054193214
2430498.91132745669312.7230567932430846.28530461669036.190145299
#Sta/Elev= 30
       0 1694.99    93.1 1695.82   118.8 1692.95   145.9  1686.9   226.4 1661.96
   262.6 1647.38   313.5 1618.89   353.5 1590.69   379.3 1562.82   412.9 1561.47
   429.6 1556.63   487.4 1558.89     843 1559.88     871 1562.71  932.311557.983
   949.2 1553.78  1094.7 1553.31  1100.5 1553.85  1107.61559.961  1117.2 1568.05
  1155.9 1591.85  1182.3 1602.51  1217.5  1605.2    1282 1616.52  1326.6  1626.1
  1343.3 1634.12  1358.6 1637.13  1387.2 1637.18  1486.5 1652.07  1639.3 1703.42
#Mann= 10 ,-1 , 0
       0      .1       0   93.53      .1       0  206.84      .1       0
  207.61      .1       0  321.69     .06       0  442.71     .05       0
  806.75    .025       0  928.09      .1       0  932.31    .045       0
  1107.6      .1       0
Bank Sta=932.31,1107.6
XS Rating Curve= 0 ,0
Exp/Cntr=0.3,0.1

Type RM Length L Ch R = 1 ,54813   ,463.8,466.4,466.9
XS GIS Cut Line= 3
2430071.24157912670529.8777747152430208.49852243670362.808555052
 2431035.1179322669438.576807708
#Sta/Elev= 30
       0 1695.14    55.6 1698.43   106.9 1696.46   237.6 1670.44     259  1661.4
   265.9  1655.5   279.6 1628.15   303.6 1603.78   314.1  1581.9   318.1 1576.22
   328.8 1570.39   350.3 1566.14     463 1560.31   527.4  1552.2   747.6 1558.04
     790 1557.14   811.8  1549.9   837.6 1550.23   914.6 1558.68 1088.19 1554.39
  1101.2 1550.32  1146.9 1549.31  1160.6 1551.18 1168.191555.259  1192.2 1574.33
  1209.2 1584.08  1314.1 1593.35  1380.6 1603.91  1419.6 1616.34  1456.2 1636.77
#Mann= 5 ,-1 , 0
       0      .1       0  392.14     .06       0   519.9      .1       0
 1088.19    .045       0 1168.19      .1       0
#XS Ineff= 2 , 0
          676.81 1571.83
Permanent Ineff=
       F       F
Bank Sta=1088.19,1168.19
XS Rating Curve= 0 ,0
Exp/Cntr=0.3,0.1

Type RM Length L Ch R = 1 ,54347   ,606.9,618.3,631.3
XS GIS Cut Line= 4
2430513.73117968670545.7025462092430781.24311185670376.395798206
2431041.61759111670111.4796613752431478.72400036669654.088187709
#Sta/Elev= 30
       0 1673.17    81.7 1668.73   114.8 1662.12   170.9 1642.56   207.2 1614.88
   237.1  1587.6   272.4 1591.71   285.2 1601.96   289.8 1602.35   321.5 1581.97
   364.4  1563.6   387.2 1557.36   471.5 1559.31   524.2 1553.32   666.6 1554.29
   755.2 1552.47  767.621548.936     777 1544.62   827.2 1544.62   847.21548.744
   887.3 1548.88   926.8 1575.34   972.2 1611.58   996.5 1613.14  1025.9 1622.79
  1083.4 1634.12  1131.5  1647.5    1224 1663.54  1297.5 1684.51  1320.7 1688.08
#Mann= 11 ,-1 , 0
       0      .1       0  176.88     .06       0  284.87      .1       0
  526.81     .05       0  552.54      .1       0  767.62    .045       0
   847.2      .1       0  875.72      .1       0  898.63      .1       0
 1036.06      .1       0 1147.64      .1       0
Bank Sta=767.62,847.2
XS Rating Curve= 0 ,0
Exp/Cntr=0.3,0.1

Type RM Length L Ch R = 1 ,53729   ,512.3,508.9,505.7
XS GIS Cut Line= 2
2430557.54244378670789.4858512882431871.65005177670320.207590371
#Sta/Elev= 30
       0 1671.35      31 1666.61      75 1653.66   141.4 1625.49   158.4 1613.66
   171.2 1609.26   183.9 1600.97   218.9 1589.75   247.6    1584   294.3 1578.15
   328.5 1578.45   349.6 1569.87     409 1558.27   675.9 1553.47   763.5 1555.88
   867.7 1554.64   951.3 1551.13   970.1  1552.3   990.9 1545.79 1058.781543.675
  1080.1 1541.31  1107.8 1541.46 1115.511545.021  1173.6  1591.6  1203.3 1617.43
    1216 1625.02  1261.1 1636.51  1305.2 1640.79    1352 1642.54  1395.4 1648.46
#Mann= 7 ,-1 , 0
       0     .05       0   60.12      .1       0   262.1     .06       0
  363.08     .05       0  969.02      .1       0 1058.78    .045       0
 1115.51      .1       0
Bank Sta=1058.78,1115.51
XS Rating Curve= 0 ,0
Exp/Cntr=0.3,0.1

Type RM Length L Ch R = 1 ,53220   ,428.8,429.9,435.7
XS GIS Cut Line= 2
 2430830.5730657671353.8361005492432143.42411453670693.549035296
#Sta/Elev= 30
       0 1667.63    68.9 1663.07    94.7 1657.19     139 1635.01   152.4 1632.43
   192.7 1609.33   210.6 1604.28     233 1586.89   267.5 1585.75   294.3 1572.22
     439    1565   474.8 1566.23   544.5    1554   582.3 1550.78   944.9 1549.01
  962.391542.254   971.8 1539.14   994.7 1539.09 1017.091542.142  1074.8 1545.16
  1110.6 1542.76  1128.3 1552.46  1191.2 1608.61  1214.8 1624.55  1267.3 1637.29
  1304.2 1631.71  1356.8 1632.42  1392.7 1643.21  1430.9 1664.84  1469.5 1680.78
#Mann= 11 ,-1 , 0
       0      .1       0   186.5     .06       0  290.63     .05       0
  394.76     .06       0  498.89     .05       0  707.15     .06       0
  770.72    .025       0  811.28     .05       0  962.39    .045       0
 1017.09     .05       0 1019.54      .1       0
Bank Sta=962.39,1017.09
XS Rating Curve= 0 ,0
Exp/Cntr=0.5,0.3

Type RM Length L Ch R = 1 ,52790   ,71.4,71.4,70
XS GIS Cut Line= 2
2431010.58714136671764.7627721282432244.09353259671110.976350039
#Sta/Elev= 30
       0 1573.45    13.8 1574.21    40.9 1572.85    86.2 1575.26   113.4 1571.34
   502.7 1564.07   511.7 1562.24   543.4 1546.92     557 1544.68   841.1 1546.53
   946.3 1545.96     969 1546.53   982.6 1550.23 1013.141543.072  1018.8 1537.14
  1023.3 1536.41  1119.9 1536.57  1125.9 1538.31 1136.791544.053  1149.5 1548.67
  1167.3 1551.86  1181.8 1549.06  1204.4 1547.92    1218 1552.62  1236.1 1551.07
  1249.7 1558.96  1300.4 1593.98  1309.3 1599.04  1322.1 1602.44  1396.1 1612.92
#Mann= 8 ,-1 , 0
       0     .06       0  174.49     .05       0  384.21     .06       0
  489.07     .05       0  908.52    .025       0 1013.14    .045       0
 1136.79    .055       0 1154.24      .1       0
#XS Ineff= 2 ,-1
       0     993 1544.82 1156.81 1396.06 1544.82
Permanent Ineff=
       F       F
Bank Sta=1013.14,1136.79
XS Rating Curve= 0 ,0
Exp/Cntr=0.5,0.3

Type RM Length L Ch R = 1 ,52718   ,385,385.5,385.6
XS GIS Cut Line= 2
2431096.74674594671805.2193841342432277.85658845671170.553986788
#Sta/Elev= 30
       0 1573.16    20.4 1571.19    61.3  1570.2   356.5 1565.48   433.7 1565.35
   443.3 1563.76   474.5 1547.97   488.1 1544.77   533.6 1544.05   792.4 1545.82
   924.1 1544.83   942.9 1542.18   957.3 1541.76  965.72 1539.43   976.7 1535.09
  1060.6  1535.1 1081.44 1539.38  1105.7 1542.59  1131.5 1541.46  1134.5 1542.36
    1142 1548.07  1145.8 1549.06  1178.4 1546.18  1199.5 1546.89  1205.4 1549.44
  1223.8 1562.16  1264.6 1593.35  1273.7 1595.52  1323.7 1600.61  1340.8 1603.96
#Mann= 9 ,-1 , 0
       0    .055       0   91.71     .05       0  301.84     .06       0
   406.9     .05       0  827.16     .06       0  965.72    .045       0
 1081.44    .055       0 1142.36     .06       0 1295.58      .1       0
Bank Sta=965.72,1081.44
XS Rating Curve= 0 ,0
Exp/Cntr=0.5,0.3

Type RM Length L Ch R = 1 ,52333   ,417.4,416,414.2
XS GIS Cut Line= 3
2431074.90558228672082.6679762152431650.17313251671940.032106623
 2432639.5891327671417.763466135
#Sta/Elev= 30
       0 1565.75      41 1568.29   201.8 1564.99   428.4 1566.42   556.2 1561.98
   589.2 1554.91   647.6 1553.31   670.2 1544.97     698 1542.57     919 1543.56
  1000.4 1541.04  1123.9 1540.92 1144.091537.443  1152.1 1532.38  1158.7 1531.78
  1231.1 1531.92 1251.981538.245  1262.7 1545.51    1266 1545.86  1301.5 1546.04
  1348.7 1542.29  1366.8 1543.25  1393.3 1548.35  1434.7 1572.95  1449.5 1575.26
  1470.2 1585.84  1520.6 1604.56  1552.2 1621.02    1611 1655.69  1711.5  1687.7
#Mann= 12 ,-1 , 0
       0    .055       0   53.52      .1       0  153.17     .05       0
  211.76      .1       0  352.48     .06       0  551.78    .055       0
  654.47     .05       0  968.87      .1       0 1144.09    .045       0
 1251.98      .1       0 1388.08     .06       0 1492.88      .1       0
Bank Sta=1144.09,1251.98
XS Rating Curve= 0 ,0
Exp/Cntr=0.3,0.1

Type RM Length L Ch R = 1 ,51917   ,358.8,353.6,353
XS GIS Cut Line= 4
2431146.70793211672743.6056307112432163.35320851 672147.98575896
2432601.43730611671898.9593541322432801.40836287671611.363800704
#Sta/Elev= 30
       0 1554.96   227.2 1552.31   266.6 1549.84     287 1554.42     328 1555.26
   348.4 1554.56   361.6 1550.52   373.3 1549.48   523.9 1545.81  1069.7 1542.22
  1255.8 1537.74  1315.6 1541.21  1366.4 1536.99    1381 1532.77 1397.631531.074
  1407.6 1527.69  1467.4 1529.28 1478.221533.121  1485.8 1539.17  1495.1 1542.92
  1545.7 1543.57  1577.1 1547.69  1591.7 1551.66  1609.9 1563.68  1633.3 1583.55
  1642.8 1588.76  1852.8 1601.35  1964.8  1627.8  1999.8 1638.14  2032.5 1651.59
#Mann= 10 ,-1 , 0
       0     .05       0  266.18     .06       0   307.6    .055       0
  414.09      .1       0  733.57     .06       0  946.56      .1       0
 1397.63    .045       0 1478.22      .1       0 1781.18     .06       0
 1915.97      .1       0
#XS Ineff= 2 , 0
          757.49 1558.52
Permanent Ineff=
       F       F
Bank Sta=1397.63,1478.22
XS Rating Curve= 0 ,0
Exp/Cntr=0.5,0.3

Type RM Length L Ch R = 1 ,51563   ,52.9,52.8,52.4
XS GIS Cut Line= 2
2431197.16714877673113.3755604622432841.70126128672165.849568382
#Sta/Elev= 30
       0  1622.1    69.1 1593.98    80.3 1588.32   105.5  1570.7   120.1 1564.16
   165.2 1553.34   237.2 1551.41   468.1 1550.67   524.3 1555.08   734.1 1545.96
     826 1545.85   865.1  1543.8  1045.7  1543.9  1107.2 1541.15  1142.1 1536.47
  1211.3 1538.92  1270.9 1536.72  1423.7 1536.29  1451.4 1530.86 1474.421531.009
  1488.3 1527.69  1589.9 1527.74 1598.291531.525  1616.8 1542.35  1622.2 1543.79
  1654.9 1542.29  1671.5 1544.28  1705.3 1571.23  1711.6 1574.64    1898 1590.15
#Mann= 14 ,-1 , 0
       0      .1       0  223.93     .05       0  494.66     .06       0
  529.16    .055       0  635.36     .06       0  765.38      .1       0
  847.75     .06       0 1036.11    .055       0 1060.14     .06       0
 1306.83      .1       0 1378.74     .06       0 1474.42    .045       0
 1598.29     .06       0 1848.28      .1       0
#XS Ineff= 2 ,-1
       0    1457 1535.22 1606.29 1897.96 1535.22
Permanent Ineff=
       F       F
Bank Sta=1474.42,1598.29
XS Rating Curve= 0 ,0
Exp/Cntr=0.5,0.3

Type RM Length L Ch R = 1 ,51511   ,432.2,435.4,438.3
XS GIS Cut Line= 2
2431274.99802986673131.9946177152432872.27337861672208.013197958
#Sta/Elev= 30
       0 1614.69    41.6 1595.48    64.4 1598.35    94.3 1593.71   129.1 1577.83
   149.9 1560.04   177.9 1552.47     240 1553.52   267.7 1549.65   420.2 1550.62
   475.7 1554.84   529.4 1548.72   668.1  1545.9   956.3 1544.65   988.6 1546.51
  1104.1  1541.5  1136.5 1535.12  1184.5 1537.91  1329.7 1536.76 1409.911530.166
  1418.4 1527.69  1524.7 1527.71 1537.731531.642  1561.6 1538.42  1619.6 1542.12
  1635.6  1551.5  1660.5 1571.38  1675.2    1576  1760.3 1587.37  1845.3 1594.53
#Mann= 12 ,-1 , 0
       0      .1       0  306.79     .05       0  450.49     .06       0
  556.76     .05       0  576.31     .06       0  981.83     .05       0
 1115.35     .06       0 1409.91    .045       0 1537.73     .06       0
 1619.43      .1       0 1654.39     .06       0 1831.97      .1       0
Bank Sta=1409.91,1537.73
XS Rating Curve= 0 ,0
Exp/Cntr=0.5,0.5

Type RM Length L Ch R = 1 ,51075   ,368,371.3,374.5
XS GIS Cut Line= 2
2431513.38797301673422.3257299662433176.76555178672559.342547789
#Sta/Elev= 30
       0 1690.31    68.3 1683.31   195.3  1616.8   213.3 1611.44   267.4 1604.54
   288.4 1594.19   303.5 1594.82   330.5 1585.38     371 1584.75   425.1 1597.61
   452.2 1575.43   469.4 1554.48   507.9 1554.56   546.8 1542.16  1196.3 1535.55
 1326.531527.581  1335.7 1525.18  1434.5 1525.08  1442.4 1529.95  1497.6 1570.97
  1533.7 1605.67  1560.7 1621.84    1579 1628.53  1602.8 1633.68  1628.3 1634.45
  1666.4 1632.72  1721.4 1622.54  1739.2 1623.03  1808.6 1633.95  1873.9 1650.94
#Mann= 14 ,-1 , 0
       0    .055       0   35.31      .1       0  139.17      .1       0
  445.14     .06       0  751.11      .1       0  767.18     .05       0
 1057.08      .1       0 1080.84     .05       0 1185.39    .045       0
 1289.95      .1       0 1326.53    .045       0  1442.4      .1       0
 1603.61     .06       0 1708.16      .1       0
#XS Ineff= 2 , 0
          693.05 1552.56
Permanent Ineff=
       F       F
Bank Sta=1326.53,1442.4
XS Rating Curve= 0 ,0
Exp/Cntr=0.3,0.1

Type RM Length L Ch R = 1 ,50704   ,424.1,434.8,441.9
XS GIS Cut Line= 3
2431783.69550326673617.6783576312432811.11864528673161.131698549
 2433287.7686106 672943.11146529
#Sta/Elev= 30
       0 1688.05   122.6  1679.2   187.2  1665.2   209.1 1655.99   231.7 1641.97
   296.6 1591.59   340.4 1569.26   352.9 1566.32   366.6 1555.96   397.3  1558.2
   546.1 1554.92   629.3 1538.57   686.5 1535.19     741  1537.4   760.6 1534.13
   808.7 1537.65  1053.8 1534.12  1084.5 1535.97  1119.5 1534.56    11641526.515
  1176.7 1523.81 1299.011526.064  1308.6  1526.7  1315.8 1530.69  1341.2 1554.35
  1374.6 1580.08  1406.4 1612.91  1431.8 1629.69  1493.4 1637.93  1648.4 1669.99
#Mann= 12 ,-1 , 0
       0      .1       0  304.59     .06       0  407.29     .05       0
  694.99     .06       0   818.1     .05       0 1068.75    .025       0
  1126.2      .1       0    1164    .045       0 1299.01      .1       0
  1332.2      .1       0 1430.27      .1       0  1435.2     .06       0
Bank Sta=1164,1299.01
XS Rating Curve= 0 ,0
Exp/Cntr=0.3,0.1

Type RM Length L Ch R = 1 ,50269   ,641.7,678.4,716.9
XS GIS Cut Line= 3
 2431824.9191741673752.9041370452432660.90962809673592.772239462
2433523.42726001673402.683380798
#Sta/Elev= 30
       0 1690.63    54.8 1685.31    83.3 1679.73     120 1669.02   254.4 1604.74
   303.2 1575.03   315.5 1572.74   356.2 1556.88   388.8 1559.02   405.1 1553.89
   441.7 1552.11   482.4 1540.76     515 1538.22   584.3 1538.66   612.8 1535.11
   816.8 1535.31   992.3 1527.61    1106 1532.39  1160.3 1527.79 1270.821524.194
  1315.9 1521.97  1356.9 1522.02 1370.731526.671  1385.5 1537.93  1422.4 1549.92
  1553.5 1615.21  1602.8 1634.11  1635.4    1651  1677.7 1666.32  1734.4 1699.08
#Mann= 11 ,-1 , 0
       0      .1       0  275.62     .06       0  374.97     .05       0
  474.33      .1       0  573.69     .06       0  673.04     .05       0
   772.4      .1       0  817.43     .05       0 1070.73      .1       0
 1270.82    .045       0 1370.73      .1       0
Bank Sta=1270.82,1370.73
XS Rating Curve= 0 ,0
Exp/Cntr=0.3,0.1

Type RM Length L Ch R = 1 ,49591   ,644.8,656.1,667.5
XS GIS Cut Line= 3
2431901.76974219673832.2763536272433013.31509128674080.273561046
2433681.94925269674338.483018383
#Sta/Elev= 30
       0 1673.35    29.7  1656.4    99.4 1603.61   132.1 1582.29   160.8 1573.99
   254.3 1558.26   297.9 1560.05   324.9 1543.88   351.5 1537.68   554.3 1529.73
   801.9 1528.85     919 1521.55   968.2 1523.57   988.1 1528.75  1161.8 1532.41
  1217.6 1524.61 1278.251523.698    1306    1519    1402 1518.59 1409.65 1525.62
  1414.8  1533.1  1449.1 1551.72  1474.9 1580.88  1496.3 1600.53  1517.7 1627.57
  1543.5 1648.42  1618.8 1720.34  1710.7 1770.21  1783.6  1799.7  1855.6 1824.15
#Mann= 7 ,-1 , 0
       0      .1       0  228.68     .06       0  335.64      .1       0
  475.83     .06       0  656.51      .1       0 1278.25    .045       0
 1409.65      .1       0
Bank Sta=1278.25,1409.65
XS Rating Curve= 0 ,0
Exp/Cntr=0.3,0.1

Type RM Length L Ch R = 1 ,48935   ,264.8,267.8,273.3
XS GIS Cut Line= 4
2432124.61969018 674278.620605292432515.80427527674514.989883214
2433143.91161487674863.6994876272433367.74614093674980.169727132
#Sta/Elev= 30
       0 1553.22    35.2 1554.25   294.4 1544.43   310.9 1539.53   334.3  1522.6
   357.7  1519.7   444.6 1519.45   469.6 1516.57   487.9  1521.4   526.8 1524.88
   702.9 1527.08   735.7 1525.08  756.39 1515.68     770 1513.34     821 1513.39
  852.181517.407   904.2 1516.45   953.4 1522.31   968.3 1527.39   986.6 1539.52
  1027.7 1576.77  1106.3  1639.5  1160.4 1653.73  1182.9  1654.4  1225.7 1638.48
  1264.3  1631.7  1309.4 1629.63  1354.5 1632.51  1399.6    1629  1427.8  1632.9
#Mann= 4 ,-1 , 0
       0     .05       0   289.7      .1       0  756.39    .045       0
  852.18      .1       0
Bank Sta=756.39,852.18
XS Rating Curve= 0 ,0
Exp/Cntr=0.3,0.1

Type RM Length L Ch R = 1 ,48667   ,348.2,347.8,348.2
XS GIS Cut Line= 3
2432086.26084301674503.7156275512433013.51226935675143.737969548
2433296.97987828675330.621125966
#Sta/Elev= 30
       0 1550.02      86 1545.31   111.9 1531.83   132.3 1525.17   331.1 1519.65
   574.9 1524.98   609.4 1523.47  635.261513.113   642.2  1511.8  743.13 1513.56
     752 1515.25   766.1  1522.4   793.4 1530.39     825 1528.72   864.7 1530.26
   876.8 1533.45   892.8 1544.54   899.7 1547.13   968.8 1553.98  1009.1 1572.85
  1040.7 1595.69  1050.4  1600.9  1118.5 1626.28  1168.8 1651.09  1214.4 1669.67
  1305.4 1700.67  1340.6 1710.05  1382.1 1720.05  1434.8  1726.1  1466.2 1734.73
#Mann= 4 ,-1 , 0
       0     .05       0   97.59      .1       0  635.26    .045       0
  743.13      .1       0
#XS Ineff= 2 , 0
                          801.42         1536.62
Permanent Ineff=
       F       F
Bank Sta=635.26,743.13
XS Rating Curve= 0 ,0
Exp/Cntr=0.5,0.3

Type RM Length L Ch R = 1 ,48319   ,47.8,48.4,49
XS GIS Cut Line= 2
 2431957.1256026674814.2143503732433113.66561237675661.893429294
#Sta/Elev= 30
       0 1548.66    13.1 1546.69    38.8 1526.65    56.6 1520.44   133.3 1520.83
   153.3 1515.43   264.9 1516.78   294.6 1519.84   433.5  1519.5   483.1 1523.01
   493.9 1521.81  507.271516.958   515.4  1511.7   522.2 1511.12     637  1511.2
  647.061515.829     657  1521.8   711.2 1518.69   788.6 1517.85   853.7 1524.09
  1033.6 1522.01  1068.3 1522.45  1083.8 1524.91  1112.9 1533.82  1167.5 1557.19
  1246.5 1609.23  1291.4 1635.78  1326.2 1649.18  1367.9 1671.56  1433.9 1700.82
#Mann= 8 ,-1 , 0
       0     .05       0    24.1      .1       0  240.51     .05       0
  507.27    .045       0  647.06    .055       0  653.82      .1       0
  791.59     .05       0 1015.06      .1       0
#XS Ineff= 3 ,-1
       0  485.27  1522.8  669.06     823  1522.8     823    1400    1530
Permanent Ineff=
       F       F       F
Bank Sta=507.27,647.06
XS Rating Curve= 0 ,0
Exp/Cntr=0.5,0.3

Type RM Length L Ch R = 1 ,48271   ,398.2,396.4,398.1
XS GIS Cut Line= 2
2431928.35827169674848.4754367172433099.73617828675718.097057045
#Sta/Elev= 30
       0 1550.19    10.8 1548.91    22.9 1541.28    37.8 1528.33    57.7 1520.44
   131.6 1520.54     195 1515.24   369.4 1520.54   486.6 1521.84   496.2 1520.22
  507.611514.269   516.1 1511.12   634.8 1511.12  643.511514.199   655.3 1520.61
   663.9  1522.5   705.4 1518.95   790.1 1516.88   818.3 1517.19   859.8 1523.53
   936.8 1521.26  1133.8 1521.59  1183.7 1535.21  1232.1  1559.4  1258.4 1575.25
  1278.3 1595.89  1298.2 1610.27    1326 1624.61  1367.3 1641.65  1458.9 1689.63
#Mann= 8 ,-1 , 0
       0     .05       0   60.79      .1       0   215.3     .05       0
  507.61    .045       0  643.51      .1       0  785.12     .05       0
 1070.03      .1       0 1430.16     .12       0
#XS Ineff= 2 ,-1
       0  237.88 1532.19  886.37 1458.89 1532.19
Permanent Ineff=
       F       F
Bank Sta=507.61,643.51
XS Rating Curve= 0 ,0
Exp/Cntr=0.5,0.3

Type RM Length L Ch R = 1 ,47874   ,405.6,406.8,403.9
XS GIS Cut Line= 3
 2431607.9947392675090.6658972052432414.08991176675707.029821962
2433167.20750001675840.724764541
#Sta/Elev= 30
       0 1556.93    27.8 1556.29    58.9 1550.41   138.7 1547.19   164.6    1541
   179.7 1531.23   199.8 1529.71   214.9 1518.34     225    1514   466.7 1517.04
   547.3 1517.06   559.31514.865   578.5 1509.56   691.8 1509.09  711.121514.736
   737.9 1519.03   874.6 1513.83   975.2 1514.31  1000.5 1515.88  1014.5 1519.74
  1109.6 1520.59  1494.8 1519.19  1531.3 1532.75  1592.3 1573.27    1641 1610.89
  1653.4 1634.14  1661.3 1644.04  1693.8 1665.08  1726.3 1676.87  1779.6 1686.19
#Mann= 9 ,-1 , 0
       0     .06       0    66.8     .05       0   559.3    .045       0
  711.12    .025       0  735.29      .1       0  742.11     .05       0
 1442.66      .1       0 1653.09     .12       0  1758.3      .1       0
Bank Sta=559.3,711.12
XS Rating Curve= 0 ,0
Exp/Cntr=0.3,0.1

Type RM Length L Ch R = 1 ,47467   ,663.1,642.4,619.8
XS GIS Cut Line= 3
2431252.07944053675358.3818972112432226.36587778676042.571473718
2433262.11413437676146.103090793
#Sta/Elev= 30
       0 1569.32    32.6 1564.01    71.7 1562.54   114.3 1552.35   315.3 1542.39
   349.7 1517.12   374.7  1510.8   622.5 1515.05  635.211511.326   651.2  1505.7
   741.3 1505.27  763.061511.199   785.3 1516.27   869.4    1516   929.7 1510.83
  1044.6 1509.25  1076.2 1520.96  1093.4 1517.37  1161.7 1516.38  1596.9 1514.28
  1834.1 1514.51  1866.3 1518.82  1906.5  1531.8  1927.5 1543.56  1950.7 1548.44
  1958.7 1557.06  2027.1  1605.5    2145 1715.78  2179.8 1738.85  2231.4 1765.52
#Mann= 12 ,-1 , 0
       0      .1       0   48.19     .05       0  146.32    .055       0
  285.06     .05       0  470.11    .025       0  562.54     .05       0
  610.75      .1       0  635.21    .045       0  763.06      .1       0
  1117.5     .05       0 1855.88      .1       0 1958.66     .12       0
Bank Sta=635.21,763.06
XS Rating Curve= 0 ,0
Exp/Cntr=0.3,0.1

Type RM Length L Ch R = 1 ,46825   ,700.2,682.5,655
XS GIS Cut Line= 3
2430785.70996645676014.9747441262431930.08300579676380.701702967
2433220.04630512  676332.0731913
#Sta/Elev= 30
       0 1609.75   135.5 1596.76   198.5  1580.8   328.6 1572.59   362.2 1562.78
     442 1554.08     499 1540.87   525.3 1529.08   530.2 1524.05  538.831508.233
   551.3 1501.88     634 1501.76     652 1501.76  674.541507.353   698.2 1511.84
     715 1507.96   769.6 1512.64  1059.3 1504.52  1095.5 1513.08  2082.7 1510.53
  2182.8 1515.69  2214.8 1527.23  2250.8  1548.2  2266.8  1552.2  2302.8 1577.19
  2322.9 1581.13  2338.9 1595.83  2384.2 1625.39  2442.9  1669.3  2492.3 1700.18
#Mann= 11 ,-1 , 0
       0    .035       0   83.32     .06       0   92.71      .1       0
  306.12     .06       0  417.52     .05       0  528.92      .1       0
  538.83    .045       0  674.54      .1       0 1183.61     .05       0
 2198.44      .1       0 2398.58     .12       0
Bank Sta=538.83,674.54
XS Rating Curve= 0 ,0
Exp/Cntr=0.3,0.1

Type RM Length L Ch R = 1 ,46143   ,792.4,782.5,762.3
XS GIS Cut Line= 2
2430745.59128028676886.8014125382433018.11265385676741.177031875
#Sta/Elev= 30
       0 1614.68    17.2  1609.2    41.2 1597.55    89.3 1578.87   253.7 1579.59
   301.8 1562.37   353.9  1557.7   361.9 1552.95     390 1529.14  415.491503.818
     434 1495.47   478.1 1495.49  531.341502.433   554.3 1507.23   570.3 1504.85
   702.6 1504.38   722.6 1505.24   734.7 1509.29     815 1507.69   934.9 1510.59
  1476.2 1509.96  1572.4 1506.68  1712.7 1508.37  2121.5 1506.12  2153.6 1511.01
  2169.6 1518.87  2193.6 1534.74  2208.4 1539.71  2225.7 1550.62  2277.2 1570.39
#Mann= 8 ,-1 , 0
       0      .1       0  154.82    .055       0  254.61    .035       0
  354.39      .1       0  415.49    .045       0  531.34      .1       0
  753.52     .05       0 2150.46      .1       0
Bank Sta=415.49,531.34
XS Rating Curve= 0 ,0
Exp/Cntr=0.3,0.1

Type RM Length L Ch R = 1 ,45360   ,673,668.9,665.1
XS GIS Cut Line= 2
2430992.09308386677750.2340688712433165.65402544677012.680097789
#Sta/Elev= 30
       0 1595.16    15.5 1584.46    32.4 1586.28    49.3 1578.38     194 1574.47
     276  1546.4   332.3 1545.18   366.1 1539.92   374.5 1536.51   391.4 1523.77
  415.871498.107   443.1  1492.5   551.9 1492.61  571.821497.222   585.7 1501.56
   691.3 1505.77   856.1 1503.62  1083.3 1506.14  1160.2 1503.95  1443.2    1505
    1684 1502.16    1836 1505.43  2000.8 1502.43  2068.3 1503.84  2089.5 1507.76
  2114.6 1519.04  2127.5 1520.75  2161.9 1536.58  2254.2 1571.24  2295.3 1590.09
#Mann= 12 ,-1 , 0
       0      .1       0  251.06    .055       0  351.77      .1       0
  415.87    .045       0  571.82    .025       0  653.89     .05       0
  754.59     .05       0  838.35     .05       0 1157.42     .05       0
 1404.99     .05       0 1660.96     .05       0 2063.79      .1       0
Bank Sta=415.87,571.82
XS Rating Curve= 0 ,0
Exp/Cntr=0.3,0.1

Type RM Length L Ch R = 1 ,44691   ,942.2,897,846.8
XS GIS Cut Line= 2
2431211.58083385678404.879085049 2433356.4476071677562.684247121
#Sta/Elev= 30
       0 1732.34    46.4 1705.89      85 1678.31    97.9 1672.68     186 1610.83
   232.3  1586.5   282.7 1567.01   299.9 1562.74   394.5 1551.64     403 1548.35
   439.1 1547.24     446 1542.99  503.191495.348   519.1 1491.13   541.7 1489.53
   609.3 1489.76  646.961494.422   673.6 1500.91   875.8 1497.59   957.4 1499.66
  1130.3 1497.63  1250.6 1500.39  1791.1 1497.35  1911.4 1501.61  2057.5 1517.86
  2114.6 1542.26  2182.5 1549.78  2212.2  1556.6  2278.1 1588.44  2304.3 1596.83
#Mann= 8 ,-1 , 0
       0      .1       0  342.09     .06       0  443.71      .1       0
  503.19    .045       0  646.96      .1       0  748.58     .05       0
 1256.69     .05       0 1991.93      .1       0
Bank Sta=503.19,646.96
XS Rating Curve= 0 ,0
Exp/Cntr=0.3,0.1

Type RM Length L Ch R = 1 ,43794   ,1047.8,1075.2,1107.9
XS GIS Cut Line= 5
2431713.48271719 679580.62443696 2432331.9476876678913.461401209
2432723.56468654678316.4281464672433273.29291779677873.870960712
2433501.19042787677738.647805959
#Sta/Elev= 30
       0  1719.5      43 1706.71   194.6 1679.68   272.5 1641.32   392.7 1567.79
   496.1  1533.1   572.6 1532.33   607.8 1526.13   984.6 1516.45    1058 1499.73
  1124.5 1499.34  1166.3 1492.88  1228.5  1495.5 1244.791490.864  1252.4 1486.41
  1285.9 1485.07 1320.581489.648  1386.4 1491.47  1415.1 1484.36  1459.6 1484.35
  1477.3 1491.01  1553.8  1496.8    1977 1494.84  2210.3 1500.14  2238.9  1506.5
  2340.5  1555.9  2391.1 1564.24  2470.7  1566.1  2498.6  1575.2  2594.5 1583.65
#Mann= 13 ,-1 , 0
       0      .1       0  538.18     .06       0  664.15     .05       0
 1064.23      .1       0 1221.64    .025       0 1244.79    .045       0
 1320.58    .025       0 1484.53      .1       0 1646.14     .05       0
 1807.27     .05       0 1874.64     .05       0 2002.32     .05       0
 2103.15      .1       0
Bank Sta=1244.79,1320.58
XS Rating Curve= 0 ,0
Exp/Cntr=0.3,0.1

Type RM Length L Ch R = 1 ,42719   ,621.9,622.4,632.2
XS GIS Cut Line= 3
2431762.25624168679764.4587149622433239.25099111679262.208735213
2434271.50876909678882.999191791
#Sta/Elev= 30
       0 1720.84   104.3 1692.18   173.7 1677.77   225.5 1672.12   262.5 1661.65
   287.8 1650.37   317.4  1631.7   414.6 1561.51     484 1519.72   520.2 1517.21
   549.8 1501.88   566.7 1498.15   963.8 1493.17    1023 1489.75  1090.6 1492.12
  1272.2 1488.41  1369.4 1493.83  1466.6 1492.82  1517.3 1486.56  1618.3 1486.67
 1704.021480.918  1717.2 1478.05  1786.6 1478.06 1799.991484.388  1840.8  1487.8
  1866.3 1504.89  2266.6 1520.31  2471.4 1540.33  2548.2 1560.51  2659.8 1609.38
#Mann= 11 ,-1 , 0
       0      .1       0  411.33     .06       0  512.04     .05       0
 1519.22     .05       0 1704.02    .045       0 1799.99      .1       0
 2227.17      .1       0 2328.33      .1       0 2429.49      .1       0
 2530.66     .12       0 2631.82      .1       0
#XS Ineff= 2 , 0
         1083.19 1505.88
Permanent Ineff=
       F       F
Bank Sta=1704.02,1799.99
XS Rating Curve= 0 ,0
Exp/Cntr=0.3,0.1

Type RM Length L Ch R = 1 ,42097   ,1367.7,1397.5,1356
XS GIS Cut Line= 4
2432081.28709969680189.9171816262433219.50627995679840.069128051
2433637.44343618679785.3074265422434228.81331643 679721.06017971
#Sta/Elev= 30
       0 1703.14    78.4 1674.44   114.5 1654.54   160.8 1621.83   252.6 1547.55
   302.8 1511.22   340.5 1508.85   369.8 1490.82   775.7 1488.21    1010  1490.2
    1077 1483.68  1212.5 1484.88  1266.7 1480.88  1290.9 1482.36 1302.11 1479.34
    1311 1473.94  1371.5 1473.92  1440.1 1474.12 1457.191479.855  1468.4 1484.68
  1492.6 1487.41  1577.3 1482.68  1698.1 1481.17  1726.2 1484.63  1754.4 1503.25
    1778 1508.72    1859 1511.26  2000.4 1524.06  2120.6 1536.28  2207.1 1548.55
#Mann= 11 ,-1 , 0
       0      .1       0  260.55     .06       0  360.81     .05       0
  561.33     .05       0  1162.9     .05       0 1262.51      .1       0
 1302.11    .045       0 1457.19      .1       0 1560.59    .045       0
    1660      .1       0 1958.36      .1       0
#XS Ineff= 2 , 0
          983.61  1495.6
Permanent Ineff=
       F       F
Bank Sta=1302.11,1457.19
XS Rating Curve= 0 ,0
Exp/Cntr=0.3,0.1

Type RM Length L Ch R = 1 ,40699   ,622.2,617.8,604.8
XS GIS Cut Line= 3
 2432340.8531816681352.0733218792433029.84064877680941.278867871
2434343.05521393 680259.28252846
#Sta/Elev= 30
       0 1808.37    72.1 1791.52   123.3 1775.64   267.7 1709.39   390.3 1629.72
     440 1591.23   454.5 1574.87   483.6 1532.68   489.5 1530.44   523.8 1528.16
   584.3 1476.01  598.62 1469.99     612 1466.53   686.8 1468.35  702.391474.565
   714.7 1478.14    1005 1475.94    1478 1476.35  1650.1 1477.41  1758.7 1480.59
  1840.1 1478.28  1893.9 1481.69  1914.1  1477.4    1948 1476.01  1964.5 1480.03
    1979 1492.87  1991.2 1499.95  2015.6 1509.21  2059.5 1516.96  2281.9  1543.8
#Mann= 8 ,-1 , 0
       0      .1       0  415.66     .06       0  545.32      .1       0
  598.62    .045       0  702.39      .1       0  842.06     .05       0
 1887.73      .1       0 2201.43     .05       0
Bank Sta=598.62,702.39
XS Rating Curve= 0 ,0
Exp/Cntr=0.3,0.1

Type RM Length L Ch R = 1 ,40081   ,508.4,506.6,504.1
XS GIS Cut Line= 2
2432705.62049669681988.2301860452434443.25448862680505.714778379
#Sta/Elev= 30
       0 1777.83    48.8 1765.28   123.8 1752.43   260.9 1722.59   369.5 1683.03
   421.7  1669.8   464.2 1654.54   511.5 1628.49   538.2 1593.76   594.7 1531.76
   637.3 1527.68   695.5 1480.72  722.771469.057   753.6 1463.88   816.5 1463.92
  842.571470.531     869 1476.78   884.8 1473.07   983.4 1471.72  1457.9 1472.96
  1524.3 1478.53  1631.5 1481.08  1873.3 1473.73  1902.7 1481.09    2002 1480.67
  2016.2 1485.12    2042 1499.94  2060.5 1502.53  2085.1 1511.47  2284.1 1533.58
#Mann= 8 ,-1 , 0
       0      .1       0  578.43     .06       0  722.77    .045       0
  842.57      .1       0   963.3     .05       0 2065.98      .1       0
 2125.14     .05       0 2251.93      .1       0
Bank Sta=722.77,842.57
XS Rating Curve= 0 ,0
Exp/Cntr=0.3,0.1

Type RM Length L Ch R = 1 ,39575   ,705.5,714,719.8
XS GIS Cut Line= 3
2433069.46819419682358.7215710432433381.08043185682092.891722128
2434819.11364502680777.430770382
#Sta/Elev= 30
       0 1712.75    30.6  1714.7     123 1731.74   166.1 1733.99   320.2 1708.22
     375 1693.49   406.6 1678.08   466.1 1629.92   485.8 1605.34   520.3 1574.39
   531.1 1557.36   547.4 1541.73   559.4 1524.75     620 1519.11   669.8 1478.53
  697.14 1467.12   731.7 1463.88  824.94 1466.47     851 1472.24  1134.2 1466.24
  1187.1 1476.55  1512.3 1475.41  1566.6 1468.82  1626.2 1473.04  1642.4  1478.7
  1756.3 1474.87  2014.7 1478.38  2048.6 1482.22  2108.1 1506.99  2358.5 1521.53
#Mann= 10 ,-1 , 0
       0      .1       0  498.22     .06       0  627.03      .1       0
  697.14    .045       0  824.94      .1       0  973.21     .05       0
 1155.53     .05       0  1210.7      .1       0 1329.45     .05       0
 1566.94     .05       0
#XS Ineff= 2 , 0
                         1643.58         1485.05
Permanent Ineff=
       F       F
Bank Sta=697.14,824.94
XS Rating Curve= 0 ,0
Exp/Cntr=0.3,0.1

Type RM Length L Ch R = 1 ,38861   ,722.2,716.1,702.4
XS GIS Cut Line= 3
2433483.54151303682844.6182370482434258.28701076  682284.1498698
2435409.14921036681333.880444884
#Sta/Elev= 30
       0 1734.97    73.1 1723.32     121 1711.22   249.9 1656.63   312.9 1619.14
   384.1 1569.25   423.6 1533.51   444.7 1509.43   494.3  1505.7     552 1467.15
   611.2 1466.69   633.51462.845   645.2 1460.46   794.2 1461.81  812.79 1466.61
   911.6 1466.57   956.8 1462.23   991.5 1469.37  1122.8 1467.29  1385.4 1471.52
  1400.7 1465.51  1420.6 1465.11    1449 1472.53  1813.3 1472.62  1911.3  1469.4
    2015 1472.47  2028.6 1475.57  2063.9 1493.51  2308.9 1514.15  2448.7 1530.58
#Mann= 12 ,-1 , 0
       0      .1       0  431.32     .06       0  548.97      .1       0
   633.5    .045       0  812.79    .025       0  860.27      .1       0
 1109.94     .05       0 1340.09     .05       0 1443.68     .05       0
 1570.24     .05       0 1634.65     .05       0 1685.31     .05       0
#XS Ineff= 2 , 0
                         1579.99         1477.51
Permanent Ineff=
       F       F
Bank Sta=633.5,812.79
XS Rating Curve= 0 ,0
Exp/Cntr=0.3,0.1

Type RM Length L Ch R = 1 ,38144   ,608.4,624.9,633.2
XS GIS Cut Line= 3
2433931.46253318683492.5355763732434681.93576977682822.289213464
2435877.23095137681700.843621716
#Sta/Elev= 30
       0 1652.75     9.8 1648.39    36.6 1651.64    68.6 1638.28     117 1634.35
   254.7 1545.19   288.6 1512.92   336.9    1509   371.7 1481.71   404.8 1465.61
   481.7 1456.69   643.7  1466.2   745.7 1466.07  786.591460.426   803.5 1456.74
     893 1456.69  918.361459.893   981.3 1454.66  1014.8 1463.54  1343.1  1466.5
  1399.7 1462.91  1473.5 1469.16  1589.3 1470.37  1923.3 1469.47  1989.1 1466.35
  2257.1 1471.78  2279.8 1474.28  2310.9 1488.62  2330.7 1492.97  2645.2 1531.02
#Mann= 16 ,-1 , 0
       0      .1       0   50.23     .06       0  180.45      .1       0
  229.62     .06       0  409.02      .1       0  769.62    .025       0
  786.59    .045       0  918.36    .025       0 1122.24      .1       0
 1125.02     .05       0 1484.26     .05       0 1963.24     .05       0
 2202.74      .1       0 2322.48      .1       0 2332.52      .1       0
 2505.41      .1       0
#XS Ineff= 2 , 0
                         1585.64         1475.44
Permanent Ineff=
       F       F
Bank Sta=786.59,918.36
XS Rating Curve= 0 ,0
Exp/Cntr=0.3,0.1
